HEC-RAS study BIGRN.prj: BIGRN

--- BIGRN.g01 (geometry) --- (continued)

Type RM Length L Ch R = 1 ,10961   ,320.1,326.8,325.7
XS GIS Cut Line= 3
 2188037.9984171657069.6036289052188057.92351066656998.618480756
2188144.23562977656656.154266246
#Sta/Elev= 30
       0 1969.59    17.1 1966.09    50.3 1955.53    62.8 1952.81    71.1 1948.77
     100 1946.43   108.2 1946.37   112.3 1945.76   120.6 1942.57   124.7 1941.87
   137.1 1941.19   149.5 1942.76     166 1943.31   190.7 1943.02     199 1943.63
   211.9 1943.68   221.5 1942.33   227.8 1941.45   236.1 1942.13   256.7  1943.2
   269.1 1942.65   281.5 1942.91   289.7 1942.38   302.1 1943.01   306.2 1943.78
   328.4 1953.81   372.2 1970.91   401.1 1981.42   410.3 1983.12   426.9 1989.18
#Mann= 4 ,-1,0
       0      .1       0      30     .06       0   221.5    .045       0
   236.1      .1       0
Bank Sta=221.5,236.1
XS Rating Curve= 0 ,0
Exp/Cntr=0.3,0.1

Type RM Length L Ch R = 1 ,10635   ,227.7,238.2,241.6
XS GIS Cut Line= 4
2188113.17348858657123.8967360842188214.24219579657037.027764598
2188269.37058154656895.0304073622188316.98146014656849.925364476
#Sta/Elev= 30
       0 1967.87    19.8 1962.99    49.4 1954.45      62 1951.63    65.5 1950.26
    69.3 1948.41    72.1  1947.5    90.1 1946.71     120 1941.47   133.3 1941.22
   150.3 1941.78   154.6 1941.65   159.4 1940.86   163.1 1940.22   165.6  1940.2
   167.4 1940.23   172.51941.035     176  1941.3   184.1 1941.15   193.2 1941.46
   202.6 1940.44   218.9 1941.87   230.5 1942.38     249 1941.97   257.5 1942.24
   270.4  1944.2   279.9 1944.59   288.3 1945.42   322.8 1947.98   351.2 1949.45
#Mann= 5 ,-1,0
       0      .1       0     120     .06       0   159.4    .045       0
   172.5     .06       0  351.18      .1       0
Bank Sta=159.4,172.5
XS Rating Curve= 0 ,0
Exp/Cntr(USF)=0,0
Exp/Cntr=0.3,0.1

Type RM Length L Ch R = 1 ,10396   ,209.8,207.6,197.8
XS GIS Cut Line= 3
2188138.02789569657275.695153545     2188297.267      657172.796
2188473.74342599657075.182464799
#Sta/Elev= 30
       0 2003.35    26.7 1992.72    56.2 1982.81    87.3 1970.12   107.5 1960.46
   121.6 1954.64   127.8 1949.55   131.1 1947.34   144.7 1945.89   153.8 1941.71
   156.7 1941.18   168.3 1940.77   174.1 1941.03   181.81940.157   188.3 1939.73
   200.3 1940.34   215.8 1940.63   229.5 1939.76   234.1 1940.14   243.2 1943.05
   247.8 1943.93   271.4 1945.62   279.7 1948.06   291.5 1950.66   298.1 1950.36
   304.5 1949.14   311.8 1949.52   326.8 1955.57   350.4 1960.08   391.3  1970.9
#Mann= 5 ,-1,0
       0      .1       0   181.8    .045       0   200.3      .1       0
  229.59     .06       0  339.59     .08       0
Bank Sta=181.8,200.3
XS Rating Curve= 0 ,0
Exp/Cntr=0.3,0.1

Type RM Length L Ch R = 1 ,10189   ,204.9,202.3,195.7
XS GIS Cut Line= 2
2188279.16399533 657487.799306762188574.64810651657145.163475706
#Sta/Elev= 30
       0 1993.53     8.7 1990.49    16.8 1988.63    29.9 1984.84    39.4  1981.4
    59.3 1975.35    82.7 1967.38   117.9 1957.59   130.2 1954.97   138.7 1949.95
   141.5 1948.96   154.7 1948.04   158.6 1947.32   167.1 1944.06     173 1941.21
   177.8 1939.94   194.21939.983   209.5 1939.45   218.1  1939.9   240.4 1939.39
   246.5  1939.6     257  1940.7   272.8 1944.09   301.7  1945.9   314.5 1948.03
   336.2 1950.64   371.3 1960.45   388.3 1965.94   422.3 1978.13   452.4 1984.74
#Mann= 4 ,-1,0
       0      .1       0   194.2    .045       0   218.1     .06       0
     330      .1       0
Bank Sta=194.2,218.1
XS Rating Curve= 0 ,0
Exp/Cntr=0.3,0.1

Type RM Length L Ch R = 1 ,9986    ,266.1,268.2,262.8
XS GIS Cut Line= 3
2188385.96393257657619.0845065912188539.60672303657512.501929598
2188675.99121451657245.377779864
#Sta/Elev= 30
       0 1979.67    36.8 1970.23    80.5 1956.35    89.2 1955.34   109.8 1954.93
   129.3 1953.19   150.7 1950.51     161 1948.33   166.8 1948.25   178.3 1949.15
   222.6 1944.92   235.6 1945.26   253.6 1943.05   271.6 1938.72   276.1 1938.19
   289.5 1938.12   311.4 1938.94   317.7 1938.21     329  1938.7   332.6 1939.42
   338.9 1942.24   343.4 1943.57   370.4 1945.77   392.8 1952.45   399.4 1953.91
   410.8 1958.28   428.8 1962.73   448.6 1969.06   469.7 1977.12   486.9 1982.82
#Mann= 5 ,-1,0
       0      .1       0     170     .06       0   311.4    .045       0
   332.6     .06       0  366.99      .1       0
Bank Sta=311.4,332.6
XS Rating Curve= 0 ,0
Exp/Cntr=0.3,0.1

Type RM Length L Ch R = 1 ,9718    ,283.9,288.6,289.6
XS GIS Cut Line= 3
2188707.52519043657711.3642934782188725.24996368657517.363044645
2188763.30154307657417.129616008
#Sta/Elev= 30
       0 1973.49    10.2 1969.02    30.3 1961.67    42.4 1957.56    50.4 1955.16
    54.4 1953.28    58.4 1950.73    62.4 1949.53    74.5 1948.81    78.5 1948.21
    86.5 1946.31    94.6 1945.16    98.6 1944.29   131.4  1940.4   136.5 1939.36
   138.8 1938.72   142.8 1938.36   146.8 1938.56   162.9 1938.98   166.9 1938.94
   174.9 1938.39   178.9 1938.44   199.3 1939.53   220.7 1939.75     225 1940.02
   237.8 1942.84   256.1 1945.76   276.3 1949.58   293.4 1951.69     302    1953
#Mann= 5 ,-1,0
       0      .1       0      80     .06       0   136.5    .045       0
   146.8     .06       0     180      .1       0
Bank Sta=136.5,146.8
XS Rating Curve= 0 ,0
Exp/Cntr=0.3,0.1

Type RM Length L Ch R = 1 ,9430    ,228.1,231.6,228.6
XS GIS Cut Line= 4
2188941.38684632657771.6208668572188960.87667966657702.014319193
2189024.91470352657492.2665888962189043.95513382657421.244357994
#Sta/Elev= 30
       0 1968.13     6.7 1966.45    19.2 1962.41    31.6 1959.14      40 1957.48
    56.5  1953.4    64.8 1951.99    77.3 1948.97    88.4 1946.73    94.8 1945.04
    98.3 1944.56   106.6 1944.33   119.2 1942.31   133.3 1941.25   144.3 1939.66
   152.6 1937.96     161 1937.51   181.9 1937.85   186.1 1937.61   194.1  1936.5
   202.8 1935.57   211.81936.432   219.5 1937.76   227.9 1939.83   240.4 1943.83
   286.5  1948.3   298.9 1950.39   311.4    1952   348.6 1962.73   365.1 1970.71
#Mann= 5 ,-1,0
       0      .1       0  142.28     .06       0   194.1    .045       0
   211.8     .06       0  242.28      .1       0
Bank Sta=194.1,211.8
XS Rating Curve= 0 ,0
Exp/Cntr=0.3,0.1

Type RM Length L Ch R = 1 ,9198    ,356.7,366.6,370.7
XS GIS Cut Line= 2
2189146.71747229657823.3889356872189246.17409185657527.725379565
#Sta/Elev= 30
       0 1964.04    31.9 1957.67    44.5 1954.57    57.2 1952.71    74.1 1951.61
    78.3 1950.76      91 1946.77    95.2 1944.92    99.4 1944.32   107.8 1944.01
   112.1 1943.55   116.3 1942.23   128.9 1937.07   132.4 1936.45   148.2 1935.85
   162.7 1937.07   170.3 1936.52   175.4 1935.76   180.2 1936.47   192.2 1939.62
   196.5 1940.32   208.2 1940.84   213.3 1941.48   217.6 1941.66     226 1941.34
   246.1 1942.23   259.8 1943.64   276.6  1946.1   306.2 1949.27   311.9 1950.18
#Mann= 5 ,-1,0
       0      .1       0     100     .06       0   170.3    .045       0
   180.2     .06       0     200      .1       0
Bank Sta=170.3,180.2
XS Rating Curve= 0 ,0
Exp/Cntr=0.3,0.1

Type RM Length L Ch R = 1 ,8831    ,120.3,137.8,150
XS GIS Cut Line= 3
2189272.48428199657836.4560387152189466.20919376657834.835543078
2189636.85660601657675.464391545
#Sta/Elev= 30
       0 1955.59    15.7 1952.63    27.7 1948.83    39.7 1946.85    55.7 1943.19
    83.7 1940.34    99.7 1939.56   115.7 1938.15   151.7 1938.53   171.7 1938.17
   193.7 1938.82   207.9 1937.42   218.9  1935.5   224.6 1935.02   241.6 1936.01
   264.2 1934.76     273 1933.81   278.4 1934.09   281.71934.909   286.9  1935.7
   309.5 1934.71   325.1 1934.97   330.9 1935.73   342.7 1938.93   349.7 1939.77
   363.3 1939.78   409.9 1942.36   415.3 1943.16   420.8  1944.7   427.2  1944.5
#Mann= 5 ,-1,0
       0      .1       0  203.73     .06       0   264.2    .045       0
   281.7     .06       0  343.73      .1       0
#XS Ineff= 2 , 0
          181.41 1942.21
Permanent Ineff=
       T       F
Bank Sta=264.2,281.7
XS Rating Curve= 0 ,0
Exp/Cntr=0.3,0.1

Type RM Length L Ch R = 1 ,8694    ,49,48.3,48.2
XS GIS Cut Line= 6
2189287.08930393657847.145696432 2189463.2021909657840.097798081
2189498.02752022 657857.212660012189589.83406538657911.998399531
 2189657.8938753658026.5533835712189713.49789171658054.619604408
#Sta/Elev= 30
       0 1954.44    21.1 1948.38    33.1 1945.91    49.1 1943.59    65.1 1942.39
    97.2 1938.39   110.7 1937.94   141.2 1938.08   180.8 1939.22   204.1 1939.39
   228.3 1936.43   240.8 1935.76   263.3 1935.97   282.8 1935.17   287.4 1934.54
   292.1 1933.82   298.3 1934.49   310.7 1934.38   315.4 1935.01     320 1936.21
   326.6  1936.7   337.3 1936.77   347.9 1935.87   353.7 1935.82   416.4 1938.36
   441.3 1941.29     461 1942.44   489.1 1946.33   497.6 1947.18   517.5 1951.75
#Mann= 5 ,-1,0
       0      .1       0   287.4    .045       0   298.3      .1       0
  351.97     .08       0  505.22     .06       0
#XS Ineff= 2 , 0
          186.93 1943.16
Permanent Ineff=
       T       F
Bank Sta=287.4,298.3
XS Rating Curve= 0 ,0
Exp/Cntr=0.3,0.1

Type RM Length L Ch R = 1 ,8645    ,187.3,183.6,173.4
XS GIS Cut Line= 6
 2189293.2400005657884.3117768772189430.12515945657878.437084535
2189475.98195305657903.9966088382189563.65663553657950.813209314
2189626.10835157658047.3783818722189693.59118781658081.806810214
#Sta/Elev= 30
       0 1959.68      23 1954.14      59  1947.2      83 1941.22      95 1939.21
   135.1 1937.73   193.5 1938.41   202.4  1937.9   216.9 1935.94     226 1935.37
   234.5 1935.68   244.1 1936.95   253.2 1935.87   258.5 1934.44   262.3 1933.77
   266.8 1933.68   276.9  1934.4   284.4 1935.47   296.5 1936.22   308.3 1935.47
   340.2 1935.22   377.8 1935.76   396.5 1936.85   403.9 1936.72   419.7 1938.58
   451.1 1940.35   460.3 1941.85   464.6 1943.59   478.1 1950.65   479.7 1950.38
#Mann= 4 ,-1,0
       0      .1       0   258.5    .045       0   276.9      .1       0
   368.9     .08       0
#XS Ineff= 2 , 0
          191.83 1942.78
Permanent Ineff=
       T       F
Bank Sta=258.5,276.9
XS Rating Curve= 0 ,0
Exp/Cntr=0.3,0.1

Type RM Length L Ch R = 1 ,8462    ,173,165.3,158.7
XS GIS Cut Line= 4
2189390.01093273658100.7222784812189461.17892231658102.185018316
2189609.27514957658101.9082069982189738.74332822658105.249321286
#Sta/Elev= 30
       0 1958.93    18.2 1952.65    26.2 1950.72    34.2 1948.07    54.8 1942.57
    62.2 1941.05    82.2 1938.13    98.2 1934.34   110.2 1934.01   130.2 1934.42
   142.2 1933.63     151 1933.83   154.2 1933.27   158.2    1933     167 1933.59
   178.2 1934.83   214.2 1934.64   222.2 1933.97   242.2 1934.05   246.2 1934.68
   254.2 1936.56   266.2 1941.23   274.2  1943.9   278.2 1944.45   290.2 1943.56
   294.2 1943.72   313.4 1945.81   318.2 1947.24   326.2 1950.88   348.8 1956.14
#Mann= 5 ,-1,0
       0      .1       0     151    .045       0     167      .1       0
  219.28     .08       0  319.28     .06       0
Bank Sta=151,167
XS Rating Curve= 0 ,0
Exp/Cntr=0.3,0.1

Type RM Length L Ch R = 1 ,8296    ,271.7,264.7,255.7
XS GIS Cut Line= 3
2189429.72938309658359.754015758     2189606.205       658251.69
2189801.75645286658133.425760383
#Sta/Elev= 30
       0 1949.78    21.6 1946.88    35.7 1945.75    54.5 1943.08    63.8 1943.29
    82.2 1941.99   110.7 1941.17   137.5 1939.08   150.5 1938.87     153  1938.6
   162.3 1935.82   171.7 1934.16   193.2 1933.23   199.9 1932.75   214.51933.166
   227.9 1934.11     242 1933.83   246.6 1934.17     256 1936.43   265.3 1937.98
   298.1 1939.59   330.8 1944.04   338.4 1945.65   361.7 1952.19   382.1 1953.06
   391.5 1954.24   396.2  1955.5   405.6  1960.9   410.2  1962.8   435.5 1967.83
#Mann= 4 ,-1,0
       0      .1       0   193.2    .045       0   214.5      .1       0
  435.47     .06       0
Bank Sta=193.2,214.5
XS Rating Curve= 0 ,0
Exp/Cntr=0.3,0.1

Type RM Length L Ch R = 1 ,8032    ,173.5,167.1,156.7
XS GIS Cut Line= 3
2189645.62259875658558.7842033292189749.77461822658492.786884061
2189880.73804864658274.170763988
#Sta/Elev= 30
       0 1950.32    20.4 1948.63      32 1946.68    50.4 1944.66    55.3 1943.98
    64.6 1941.68    69.3 1940.97    88.3  1939.2   100.1 1939.08   111.9 1937.19
   121.4 1936.87   133.5 1933.68   135.8  1933.4   160.1 1933.61   169.5  1932.3
   182.5 1931.35   191.8 1931.84   194.7 1932.68     198 1933.57   211.4 1933.44
   230.1 1935.02   244.3 1937.58   258.1 1939.07   302.6 1946.24   322.6 1948.26
   346.4 1952.34     356 1955.01   363.9 1958.93   366.8 1959.85   378.1 1960.68
#Mann= 3 ,-1,0
       0      .1       0   169.5    .045       0   194.7      .1       0
Bank Sta=169.5,194.7
XS Rating Curve= 0 ,0
Exp/Cntr(USF)=0,0
Exp/Cntr=0.3,0.1

Type RM Length L Ch R = 1 ,7864    ,337.9,354.9,365.2
XS GIS Cut Line= 3
2189884.00979331658635.1840218692189900.71536475658500.704171781
2189974.21987909658396.294350284
#Sta/Elev= 30
       0 1937.83    10.1 1937.27    22.2  1937.6    30.2 1937.61    34.3 1937.99
    38.3 1937.97    50.4 1937.14    62.5 1935.65    74.6 1933.78    78.6 1932.51
    82.6 1931.45    90.7 1930.89    98.8 1931.34   105.9 1932.21   114.9 1933.42
   122.9    1934     131 1935.12   139.8 1935.33   144.7  1935.9     175 1937.58
   183.2 1938.45   190.2 1939.69   197.1 1941.19   206.6 1942.66   213.2 1943.91
     223 1945.12   242.6  1949.8   252.3 1953.04   258.2 1954.04   263.2 1954.18
#Mann= 3 ,-1,0
       0      .1       0    78.6    .045       0   105.9      .1       0
Bank Sta=78.6,105.9
XS Rating Curve= 0 ,0
Exp/Cntr(USF)=0,0
Exp/Cntr=0.3,0.1

Type RM Length L Ch R = 1 ,7510    ,194,202.6,207.8
XS GIS Cut Line= 4
2189998.25734022658679.6394036452190058.67582359658655.230707597
2190205.25433974658608.2877048442190282.43767215658591.749536127
#Sta/Elev= 30
       0 1935.42    12.6 1935.47      31 1933.93    40.9 1934.11    58.2  1933.6
    70.9 1933.74    87.7 1934.76    96.1 1934.76   112.9  1932.9   125.5 1930.73
   154.9 1931.12   163.7 1930.56   171.7 1929.66   176.8 1931.16   188.9 1936.08
   192.1 1936.67   201.1 1937.34   204.8 1938.49   209.5 1942.14   213.7 1944.96
   230.2 1953.53     241  1957.3   250.7 1961.18   258.9 1963.81   267.1  1967.3
   271.3  1968.3   283.4 1968.78   287.5  1969.5   294.9 1974.21     298 1975.59
#Mann= 3 ,-1,0
       0      .1       0   163.7    .045       0   176.8      .1       0
Bank Sta=163.7,176.8
XS Rating Curve= 0 ,0
Exp/Cntr(USF)=0,0
Exp/Cntr=0.3,0.1

Type RM Length L Ch R = 1 ,7307    ,338.6,319.5,284.7
XS GIS Cut Line= 3
2190023.57091964658780.4673688582190174.16183305 658818.73195842
2190257.34865198658841.375629101
#Sta/Elev= 30
       0 1933.72     4.4  1933.5    17.1 1933.51    41.9 1932.03    50.1 1932.42
      79 1931.48    87.3 1930.86    95.5 1929.44   103.8  1928.6   107.9 1928.93
   112.1 1929.57   124.4 1929.86   128.6 1929.57   132.6 1928.14   136.8 1926.69
   140.9 1926.45   149.2 1928.37   153.3 1929.23   157.5  1929.5   169.9 1929.03
     174 1929.48   178.6 1931.01   182.3 1932.88   186.5 1933.71   191.6 1933.57
   203.1  1935.1   223.8 1937.17   227.9 1937.73     234 1937.86   241.6 1938.36
#Mann= 3 ,-1,0
       0      .1       0   132.6    .045       0   149.2      .1       0
Bank Sta=132.6,149.2
XS Rating Curve= 0 ,0
Exp/Cntr(USF)=0,0
Exp/Cntr=0.3,0.1

Type RM Length L Ch R = 1 ,6988    ,135.5,135.5,135.2
XS GIS Cut Line= 3
2190150.37106027659161.8200180932190164.22693799659012.402264514
2190174.42708314658961.102577246
#Sta/Elev= 30
       0  1931.8     4.7 1931.57     8.7 1931.09    16.7 1930.64    28.8 1929.49
    36.8 1928.93    56.9  1926.8    64.9 1926.83    68.9 1926.63      77 1925.45
      85 1925.16      93 1925.14    97.1 1924.63   101.5 1922.95   103.9 1922.27
   105.1 1921.93   113.1 1921.24   117.1 1921.27   125.2 1922.01   129.2 1922.86
   133.2  1924.3   137.2 1925.38   145.6 1926.54   161.5    1928   165.6 1928.15
   177.8  1927.9     186 1928.25   190.8 1927.99   198.2 1928.01   202.4 1927.82
#Mann= 3 ,-1,0
       0      .1       0   103.9    .045       0   125.2      .1       0
Bank Sta=103.9,125.2
XS Rating Curve= 0 ,0
Exp/Cntr(USF)=0,0
Exp/Cntr=0.3,0.1

Type RM Length L Ch R = 1 ,6852    ,155.7,172.9,184.8
XS GIS Cut Line= 3
 2190266.4319803659162.7149946992190289.38866179 659137.58342881
2190300.70856495658997.731081541
#Sta/Elev= 30
       0 1923.64     2.6 1923.86     7.5 1923.86    12.9 1922.95    16.5 1922.64
    22.1 1922.73    30.6 1923.17    34.4 1923.14    42.5 1922.72    62.5 1922.37
    74.1  1922.9    78.6 1922.91    82.6 1922.26    94.6 1919.75    98.7  1919.1
   101.3 1918.81   106.7 1918.22   110.7 1918.05     115 1918.12   118.8 1918.41
   122.7 1918.57   126.7 1919.16   134.8 1922.17   138.8 1923.28   142.8 1924.09
   144.7 1924.59   154.8  1927.5   163.2 1929.25   170.7 1930.66   174.3 1930.96
#Mann= 3 ,-1,0
       0      .1       0   101.3    .045       0   126.7      .1       0
Bank Sta=101.3,126.7
XS Rating Curve= 0 ,0
Exp/Cntr(USF)=0,0
Exp/Cntr=0.3,0.1

Type RM Length L Ch R = 1 ,6679    ,171.8,164.8,158.4
XS GIS Cut Line= 3
2190289.50508519659207.8913011142190431.89474556659123.370820866
2190463.26860212659111.196978721
#Sta/Elev= 30
       0 1922.65    12.4 1922.74    18.5 1921.86    26.4 1921.22    35.7 1919.75
    44.8 1918.77    49.6 1918.87    54.3 1919.61    58.9 1919.81    63.6 1918.84
    68.2 1918.53    94.4 1918.59   114.7 1919.67     124 1920.46   128.7 1920.17
   130.7 1919.76   133.3 1918.99     138  1917.1   142.7 1916.05     147 1916.53
   149.9 1917.23     162 1920.39   165.9 1920.21   170.6 1920.69   174.5 1922.39
   179.9 1926.66     183  1929.4   187.3 1932.71   195.3 1935.89   199.2 1937.82
#Mann= 3 ,-1,0
       0      .1       0     138    .045       0   149.9      .1       0
Bank Sta=138,149.9
XS Rating Curve= 0 ,0
Exp/Cntr(USF)=0,0
Exp/Cntr=0.3,0.1

Type RM Length L Ch R = 1 ,6514    ,123.2,133,141.5
XS GIS Cut Line= 4
2190393.92057591659332.6440709272190425.98011277659312.915125169
2190470.37024073659251.2621696722190510.32135589659209.831383579
#Sta/Elev= 30
       0 1921.26     4.2 1921.02    12.9 1920.91    21.4 1920.58    30.8 1920.67
    35.5 1920.56    48.2  1919.5    52.1 1918.98      57 1917.55      62  1915.1
    64.8 1913.99    66.9 1913.24    68.8 1912.92    71.8 1912.64    76.7 1912.84
    82.5 1913.51    86.6    1914    96.3 1914.91   101.4 1915.17   109.9 1916.02
   113.6 1916.21     122 1916.87   127.7 1916.72   133.2 1916.99   139.3 1918.48
     145 1920.79   150.8 1922.74   155.4 1923.96   161.6  1925.4   171.2 1927.39
#Mann= 3 ,-1,0
       0      .1       0    64.8    .045       0    82.5      .1       0
Bank Sta=64.8,82.5
XS Rating Curve= 0 ,0
Exp/Cntr(USF)=0,0
Exp/Cntr=0.3,0.1

Type RM Length L Ch R = 1 ,6381    ,136.7,146.8,155.7
XS GIS Cut Line= 4
2190452.86835646659375.4672496952190531.29091585659347.846725633
2190581.59972753659338.4754763972190639.80011752 659325.15843801
#Sta/Elev= 30
       0 1919.77    16.2 1919.48    24.7 1918.61    37.4 1918.07      42 1917.69
    48.3 1916.73    57.7 1914.45    60.8 1914.05    67.1 1913.81    71.4  1913.8
    75.6 1913.98    79.1 1913.88      84 1913.28    97.7 1912.66   104.4 1912.22
   112.5 1911.54   116.6 1912.05   118.81912.514   124.7 1913.52   141.1 1915.04
   145.2 1915.59   149.3 1917.25   153.4 1919.21   161.6 1922.67   169.8 1926.36
   173.9 1927.91   182.1 1929.55   186.2 1930.79   190.3 1932.44     194 1933.22
#Mann= 3 ,-1,0
       0      .1       0   104.4    .045       0   118.8      .1       0
Bank Sta=104.4,118.8
XS Rating Curve= 0 ,0
Exp/Cntr(USF)=0,0
Exp/Cntr=0.3,0.1

Type RM Length L Ch R = 1 ,6235    ,162.2,147.8,127.8
XS GIS Cut Line= 3
 2190440.9570286659435.786171632 2190517.9747884659485.944796717
2190553.24762798659501.801394325
#Sta/Elev= 30
       0 1918.87     3.8  1918.7    20.7 1918.49    22.9 1918.37    27.7  1917.6
    31.9 1916.85      38 1915.21    39.2 1915.03    40.9 1914.44    46.5 1912.86
    52.5    1910    56.3 1908.84    61.2 1908.31    66.9 1908.07    70.7  1908.2
    74.7 1908.79    75.6 1908.95    80.2 1910.33      85  1911.4    90.5 1911.88
      96 1912.05   103.1 1912.06   107.5 1912.42   111.9 1914.09   116.3 1916.42
   119.3 1917.34   120.6 1917.61   126.3 1917.17   129.4 1916.66   130.6  1916.8
#Mann= 3 ,-1,0
       0      .1       0    56.3    .045       0    74.7      .1       0
Bank Sta=56.3,74.7
XS Rating Curve= 0 ,0
Exp/Cntr(USF)=0,0
Exp/Cntr=0.3,0.1

Type RM Length L Ch R = 1 ,6087    ,150.6,152.3,152
XS GIS Cut Line= 4
2190417.25862168659639.3560882582190478.78333903659599.804484248
2190494.76378509659588.6181720022190566.67579238659541.475856112
#Sta/Elev= 30
       0  1923.7     8.2 1924.11    11.4 1923.83      13 1923.54    18.8 1921.87
    27.2 1920.54      32 1918.81    38.4  1915.5    44.2 1911.71    48.4 1908.28
      50 1907.41    52.9 1906.58    55.8 1906.25    58.7 1906.24    63.2 1906.47
    70.3 1907.38    77.7 1908.39    90.4 1909.81      99 1909.78   108.7 1909.11
     123 1908.85   139.5 1909.57   142.4 1909.88   145.3 1910.83   151.7 1913.96
   156.8  1915.5   161.3 1916.22   165.5 1916.65   171.9 1916.49   178.6  1916.9
#Mann= 3 ,-1,0
       0      .1       0      50    .045       0    70.3      .1       0
Bank Sta=50,70.3
XS Rating Curve= 0 ,0
Exp/Cntr(USF)=0,0
Exp/Cntr=0.3,0.1

Type RM Length L Ch R = 1 ,5934    ,165.9,168.8,168.9
XS GIS Cut Line= 3
 2190516.9056364659695.0384869722190570.61769122659670.180015316
2190650.07602027659646.653247498
#Sta/Elev= 30
       0 1915.97     6.9  1915.5      14 1914.77    21.2  1914.2      25 1913.68
      28 1912.88    34.5 1910.78    43.3 1907.54      46 1907.09    47.7 1906.93
      52 1906.84    60.8 1906.18      65 1906.06    69.2 1905.58    77.3 1903.72
    81.7 1902.85    85.8 1902.51      87 1902.65    90.9 1903.49    94.2 1904.62
    98.4 1906.94   102.5 1909.47     105 1910.55   106.7 1911.16   110.9 1912.26
     115 1913.11   119.2 1913.78   131.7 1915.06   138.5 1915.32   142.1 1915.33
#Mann= 3 ,-1,0
       0      .1       0    77.3    .045       0    90.9      .1       0
Bank Sta=77.3,90.9
XS Rating Curve= 0 ,0
Exp/Cntr(USF)=0,0
Exp/Cntr=0.3,0.1

Type RM Length L Ch R = 1 ,5766    ,191.5,194.7,195.8
XS GIS Cut Line= 4
2190575.99681264659826.2427352582190624.73717314659818.252512226
2190666.68584406  659811.86033382190705.43842577659806.267177677
#Sta/Elev= 27
       0 1906.51     4.2 1906.27     8.3 1906.27    12.3 1906.11    16.4 1905.76
    24.5 1906.02    28.6 1905.99    36.7 1905.33    40.7 1904.37    48.8 1902.23
    52.9 1900.48    56.41898.507    56.9 1898.22      61  1897.1      65 1897.27
    69.1 1898.08      711898.531    77.1 1899.99    83.1  1901.1    85.2 1901.46
    93.3 1902.48   101.4 1903.75   105.5 1904.61   109.5 1905.29   116.7 1906.07
   120.2 1906.11     131 1905.99
#Mann= 3 ,-1,0
       0      .1       0    56.4    .045       0      71      .1       0
Bank Sta=56.4,71
XS Rating Curve= 0 ,0
Exp/Cntr(USF)=0,0
Exp/Cntr=0.3,0.1

Type RM Length L Ch R = 1 ,5571    ,111.3,112.8,113.4
XS GIS Cut Line= 3
2190526.20583166660005.9216392552190710.86876396660005.477737976
2190941.69742934660018.350875083
#Sta/Elev= 30
       0  1903.2      10 1901.81      18 1901.09      34 1898.65      58 1896.42
      78 1898.04      90 1897.66      98 1898.01     102 1897.78     118 1893.99
     126 1892.82     134 1891.58   146.4  1892.7     150 1892.68     170 1894.67
   177.7 1894.99     194 1894.42     202 1894.56   242.1  1893.6   262.7 1892.73
   271.2 1893.03   282.1 1892.63   302.2 1893.12   326.2 1895.62   342.2 1896.79
   362.2  1897.1   370.3 1897.67   386.3 1900.06   394.3 1900.72   415.9 1903.51
#Mann= 3 ,-1,0
       0      .1       0     126    .045       0   146.4      .1       0
Bank Sta=126,146.4
XS Rating Curve= 0 ,0
Exp/Cntr(USF)=0,0
Exp/Cntr=0.3,0.1

Type RM Length L Ch R = 1 ,5458    ,278.5,277.1,276.6
XS GIS Cut Line= 3
2190419.10176192660101.6417620432190698.45603988660120.203508086
 2190875.7207146660223.221198629
#Sta/Elev= 30
       0 1910.23    53.2 1897.94    93.3 1894.67   105.3 1891.86   109.3 1891.51
   113.3  1891.5   121.3 1893.34   137.4 1895.07   153.4 1895.37   169.4 1893.12
   177.5 1892.68   193.5 1893.32   218.6 1893.32   222.4 1892.95   229.6 1890.61
   237.4  1888.7   241.6 1888.54   250.7 1890.23   265.7 1892.97   273.7 1893.35
   300.5 1892.64   328.2 1889.75   351.4 1889.44   363.9 1889.99   369.9 1890.53
   383.7 1893.63   397.6 1895.44     430 1897.89     457 1903.25     485 1908.13
#Mann= 3 ,-1,0
       0      .1       0   229.6    .045       0   250.7      .1       0
Bank Sta=229.6,250.7
XS Rating Curve= 0 ,0
Exp/Cntr=0.3,0.1

Type RM Length L Ch R = 1 ,5181    ,236.3,249.6,252.6
XS GIS Cut Line= 4
2190361.56034919660237.1425081622190455.29716671 660257.56042881
 2190537.8969366660277.0502621562190678.96620654660403.270135254
#Sta/Elev= 30
       0 1910.05    19.1 1906.47    27.2 1905.23    43.6 1903.98    76.4 1898.51
    89.6 1897.62    96.8 1896.78   109.6 1894.81   121.5 1892.27   132.9 1887.77
   137.9 1886.81   154.4 1886.04   158.5 1886.14   163.9 1887.26   174.9 1890.08
     179 1890.36     199 1889.94   210.7 1890.25   219.3 1889.76     229 1890.49
   248.3 1889.71   264.4 1890.69     276 1892.66   291.2 1893.86   307.3 1894.17
   321.3 1893.82   335.5 1894.51   350.2 1896.22     361 1898.47   370.1  1899.9
#Mann= 3 ,-1,0
       0      .1       0   132.9    .045       0   163.9      .1       0
Bank Sta=132.9,163.9
XS Rating Curve= 0 ,0
Exp/Cntr=0.3,0.1

Type RM Length L Ch R = 1 ,4931    ,208.3,183,157.6
XS GIS Cut Line= 3
2190408.20418374660276.7589776922190536.83708382660417.921056354
2190604.49464815 660547.38923501
#Sta/Elev= 30
       0 1902.04    11.8  1899.5      33 1896.21    42.7 1895.74    53.4 1894.29
    70.9 1893.11    76.3 1892.38    82.4 1891.03    93.7 1889.47      98 1889.35
   106.9 1889.96   124.9 1889.38   136.5 1889.51   146.7    1889   154.4 1889.19
   162.9 1888.47   184.3 1888.24     190 1887.81   206.8 1888.38   230.8 1885.33
   241.4  1883.9   244.3 1884.17   248.61885.417   253.3 1887.04   261.1  1889.1
     270 1892.69   275.9 1894.44   289.4 1895.42   325.5 1900.32   337.1 1900.79
#Mann= 3 ,-1,0
       0      .1       0   230.8    .045       0   248.6      .1       0
Bank Sta=230.8,248.6
XS Rating Curve= 0 ,0
Exp/Cntr(USF)=0,0
Exp/Cntr=0.3,0.1

Type RM Length L Ch R = 1 ,4748    ,122.3,123.1,124
XS GIS Cut Line= 3
2190253.95360179660546.9758464512190462.25764073660495.415440774
2190553.00395472660546.975846451
#Sta/Elev= 30
       0 1903.66    10.5 1901.53    24.1 1899.54    35.3 1897.93    43.5 1897.31
    57.4 1894.85    76.5 1892.12   101.2 1889.01   105.3 1888.98   115.6 1889.86
   125.9 1891.55   135.4 1891.57   138.3 1891.21   142.4 1890.09   150.6 1886.54
   155.3 1884.86   158.9 1883.92   168.5  1883.5   178.4 1883.69   183.6 1884.41
   191.8 1886.24     196 1886.81   204.8 1887.23   230.6 1887.71   249.6 1889.96
   258.4 1890.52     273 1892.46   281.8 1893.28   290.4 1893.69     319 1894.17
#Mann= 3 ,-1,0
       0      .1       0   155.3    .045       0   183.6      .1       0
Bank Sta=155.3,183.6
XS Rating Curve= 0 ,0
Exp/Cntr(USF)=0,0
Exp/Cntr=0.3,0.1

Type RM Length L Ch R = 1 ,4625    ,159.3,176.3,188.2
XS GIS Cut Line= 3
2190282.87344119660607.2394081332190433.22358415 660623.01689227
2190566.86815566660592.390011298
#Sta/Elev= 30
       0 1900.16    24.8 1896.22    29.5  1895.6    37.5 1895.12    53.6 1892.56
    65.7  1889.7    73.7 1886.13    77.7 1885.26    85.8 1885.17   101.9 1885.77
   109.9 1886.33     122 1887.93   162.4 1887.81   166.5 1887.67   170.6 1886.98
   181.9 1883.09     187 1882.22   201.9 1881.62   207.6 1882.02   211.7 1882.71
   213.1 1883.21   215.8  1884.2     224 1888.13   228.6 1889.92   232.2 1891.19
   236.3 1891.96   244.5 1893.01   265.3 1894.02   281.4 1895.63   288.3 1897.02
#Mann= 3 ,-1,0
       0      .1       0   181.9    .045       0   213.1      .1       0
Bank Sta=181.9,213.1
XS Rating Curve= 0 ,0
Exp/Cntr(USF)=0,0
Exp/Cntr=0.3,0.1

Type RM Length L Ch R = 1 ,4449    ,209.7,214.4,220.7
XS GIS Cut Line= 3
2190273.56790556660705.215176658 2190405.6461836 660735.15062521
2190548.03209152660819.706810518
#Sta/Elev= 30
       0  1894.4    12.2 1893.36    27.3 1892.48    54.1 1891.76    72.4 1891.63
   105.2 1892.12   109.1 1891.93   129.8 1886.11   133.9 1885.41     143    1885
   152.8 1883.45   159.2  1882.8   167.9 1883.17   171.2 1883.71   175.6 1884.62
   194.2 1890.17   203.5  1892.4   208.2  1893.2   217.7 1894.29   226.3 1894.41
   236.1 1895.01   240.7 1895.03   245.4 1895.69   256.9 1898.11   273.3 1901.22
   277.9  1902.5   287.6  1906.4   290.5 1907.19   293.5 1907.59     301 1907.98
#Mann= 3 ,-1,0
       0      .1       0   152.8    .045       0   171.2      .1       0
Bank Sta=152.8,171.2
XS Rating Curve= 0 ,0
Exp/Cntr=0.3,0.1

Type RM Length L Ch R = 1 ,4235    ,273,246.8,228.7
XS GIS Cut Line= 4
2190214.41983621660816.4841820422190332.28692358660888.874991613
2190396.32494743660987.2522456442190425.82895735661028.844306224
#Sta/Elev= 30
       0 1891.75     7.6 1890.48    13.4 1889.95    30.2 1889.26    62.5 1888.47
    83.2 1886.72   100.7 1884.56   109.4  1883.8     121 1883.58   147.1 1884.38
   176.9 1882.72   181.6 1881.77   187.6 1878.84   191.2 1877.23   193.4 1877.08
     196 1877.12   204.1    1879   216.5 1881.67   222.3 1883.52   225.2 1884.87
   234.1 1890.53   238.9 1893.15   243.7 1894.35   248.5 1894.93   253.2 1894.44
   258.1 1893.38   272.8  1892.6   279.9 1894.71   294.3 1896.92   306.7 1899.81
#Mann= 4 ,-1,0
       0      .1       0  138.32     .06       0   187.6    .045       0
   204.1     .06       0
Bank Sta=187.6,204.1
XS Rating Curve= 0 ,0
Exp/Cntr=0.3,0.1

Type RM Length L Ch R = 1 ,3988    ,129.8,118.8,109.7
XS GIS Cut Line= 3
 2189969.8058138661027.6985194312190196.46754339661044.077354741
2190375.41433846661057.488976045
#Sta/Elev= 30
       0 1896.07    46.5  1892.9    66.5 1892.69    78.6 1891.81   114.7  1891.4
   122.7 1889.69   134.7 1888.89   138.7 1887.68   150.8 1880.56   154.8 1879.01
   165.2 1877.03   170.8 1875.98   186.9 1875.34   194.9 1875.89   199.8 1877.19
   202.9 1878.71   206.9 1881.31   210.9 1882.64   222.9  1882.5     231    1883
     243 1882.94     259 1884.39   283.1 1888.65   290.8 1889.47   307.2 1890.24
   351.3 1890.13   375.4 1891.08   392.2 1890.07   395.4  1890.4   406.7 1896.08
#Mann= 4 ,-1,0
       0     .06       0      30      .1       0   165.2    .045       0
   199.8      .1       0
Bank Sta=165.2,199.8
XS Rating Curve= 0 ,0
Exp/Cntr=0.3,0.1

Type RM Length L Ch R = 1 ,3869    ,150.7,143.8,134.1
XS GIS Cut Line= 3
2190040.10563949661223.0790813892190249.76056106661118.669259892
2190328.27674682661097.787295593
#Sta/Elev= 30
       0 1899.17     4.3 1898.71       9 1897.52      18 1894.44    26.9 1892.82
    73.1 1888.75    99.9 1887.22   102.9 1886.75   107.3 1885.29   116.3 1883.01
   125.2 1879.77   129.7 1879.18   138.6 1878.96   144.7  1877.1   147.5 1876.14
   153.6 1875.28   156.5  1875.4   162.6    1877   174.5 1879.27   192.2 1878.41
   196.7 1878.79   205.6 1881.43     219 1886.74   223.5 1888.12   228.2 1888.94
   236.7 1889.29     257 1889.16     274 1889.58   298.8 1889.38   315.5 1889.83
#Mann= 4 ,-1,0
       0     .06       0     100      .1       0   144.7    .045       0
   162.6      .1       0
Bank Sta=144.7,162.6
XS Rating Curve= 0 ,0
Exp/Cntr=0.3,0.1

Type RM Length L Ch R = 1 ,3725    ,73.9,73.1,77.4
XS GIS Cut Line= 4
2190201.22459841661506.5224330692190265.68118714661265.209939815
2190308.80875357661207.0378734752190381.02235316661129.809440574
#Sta/Elev= 30
       0 1901.28     9.7 1900.92    13.3 1900.15      18 1898.14    26.2 1893.76
    29.6 1893.02    52.5 1893.23    71.8 1892.67    80.1 1892.04   111.3 1888.43
   140.7 1887.66   162.9 1887.64   181.9  1886.6   212.6 1883.93   249.8 1878.46
   265.9 1877.95   274.1 1876.71   280.8 1875.75   294.3 1875.07     301 1876.66
   314.5  1883.6   319.5 1884.24   335.7  1884.4   350.5 1885.45     374 1885.12
   379.8 1885.98   391.5 1892.77   393.8 1893.36   419.3 1897.13   427.9 1898.77
#Mann= 4 ,-1,0
       0     .06       0   274.1    .045       0     301     .06       0
  362.19      .1       0
Bank Sta=274.1,301
XS Rating Curve= 0 ,0
Exp/Cntr=0.3,0.1

Type RM Length L Ch R = 1 ,3652    ,87.9,105.2,115.2
XS GIS Cut Line= 5
2190248.06625418 661516.316093192190287.88027953661334.325596047
2190329.18920892 661288.240746492190356.72339963661243.340321979
2190413.11728632661162.907340389
#Sta/Elev= 30
       0 1892.53    16.2 1890.67    29.6 1887.05      36 1885.73    44.2  1885.3
    56.4 1883.86    75.4 1882.98   138.3 1882.89   150.7 1882.62   175.2 1881.12
   201.5 1880.05   204.7 1879.67   210.7 1877.69   216.7 1876.28   225.4 1876.32
   230.8 1875.92   241.6  1877.2   246.7 1877.57   253.9 1878.73   265.9 1881.54
   275.2 1882.07   284.6  1883.2   289.3 1884.44   298.7 1887.79   307.8 1891.74
   313.8 1893.82     325 1895.45   344.6 1898.91   371.9  1902.7   399.1 1907.75
#Mann= 3 ,-1,0
       0     .06       0   210.7    .045       0   241.6     .06       0
Bank Sta=210.7,241.6
XS Rating Curve= 0 ,0
Exp/Cntr=0.3,0.1

Type RM Length L Ch R = 1 ,3547    ,133.1,135,135.9
XS GIS Cut Line= 4
2190255.37458637 661527.677908622190302.70481137661396.458317856
2190401.83817813661384.080742337 2190502.4570043661372.606771177
#Sta/Elev= 30
       0 1892.58     6.9 1890.97    15.4 1889.37    19.7 1887.97    28.2 1884.51
    46.3 1880.79    49.4 1880.54    74.9 1880.75   113.2 1881.54   139.5 1881.15
   157.1 1879.62   169.2 1879.94   189.3 1876.93   201.4 1875.19   205.5 1875.02
   215.4 1877.09   221.6 1878.97   226.2 1881.52   229.5 1883.79   233.7 1886.05
   240.5  1888.3   245.8 1889.41   265.8 1892.62   293.3 1898.19     302 1900.37
   310.2 1903.25   314.2 1904.04   322.3    1905   334.3 1909.41   340.7 1910.68
#Mann= 4 ,-1,0
       0     .06       0     110      .1       0   189.3    .045       0
   215.4      .1       0
Bank Sta=189.3,215.4
XS Rating Curve= 0 ,0
Exp/Cntr=0.3,0.1

Type RM Length L Ch R = 1 ,3412    ,197.4,176.6,158.3
XS GIS Cut Line= 3
2190262.94396432661584.7245116112190319.39067024661523.345569251
2190448.17684394661504.712676035
#Sta/Elev= 30
       0 1895.72    11.9 1893.58    21.1 1893.35    31.4 1892.17    37.4 1891.83
    42.9 1890.79    49.1 1888.73    59.2  1883.4    64.6 1880.92    71.3 1878.67
    78.6 1876.85    84.2 1876.93    96.3 1879.04   100.3  1878.2   104.4 1876.67
   108.4 1875.56   112.5 1875.06   116.5 1875.17   121.3  1876.6   128.6 1878.52
   144.8 1880.25   152.9 1882.18     161 1883.41   169.1 1885.94   173.1 1886.57
   181.2 1886.83   201.4 1890.27   205.4 1891.23   209.5 1892.83   213.5 1893.55
#Mann= 6 ,-1,0
       0     .08       0      20     .06       0      50     .07       0
   104.4    .045       0   121.3     .07       0  163.39      .1       0
Bank Sta=104.4,121.3
XS Rating Curve= 0 ,0
Exp/Cntr(USF)=0,0
Exp/Cntr=0.3,0.1

Type RM Length L Ch R = 1 ,3235    ,107.1,147.7,168.3
XS GIS Cut Line= 4
2190412.55513632661690.493581927 2190460.2334219661637.335033633
 2190460.2334219661552.9389878892190473.38605241661515.125175185
#Sta/Elev= 30
       0 1882.73     7.1 1882.86    11.4 1882.34    23.3 1879.62    29.4 1877.88
    35.4 1876.87    50.1 1875.79    59.3 1874.55    65.3 1874.06    79.6 1874.47
    83.6 1873.94    91.6 1872.19    99.6  1871.5   103.6  1871.5   107.6 1871.81
   110.11872.361   115.5 1873.47   119.6 1873.45   131.6 1871.93   135.6 1871.85
   139.6 1872.91   143.6 1875.07   151.6 1880.01   155.5  1882.1     164 1886.49
   168.3  1888.1   171.3 1888.82   176.7 1890.53   183.8  1892.2   195.8  1893.5
#Mann= 4 ,-1,0
       0     .12       0    91.6    .045       0   110.1     .12       0
  141.41      .1       0
Bank Sta=91.6,110.1
XS Rating Curve= 0 ,0
Exp/Cntr=0.3,0.1

Type RM Length L Ch R = 1 ,3088    ,138.4,132.6,123.8
XS GIS Cut Line= 3
2190407.28511322661717.2401206082190466.22410238 661687.26702283
2190623.81765736661688.594393914
#Sta/Elev= 30
       0 1881.76     5.5 1881.84    15.6 1880.57    27.9 1880.23    35.4 1879.65
    45.9  1877.5    54.8 1875.17    59.3 1874.42      70 1873.21    80.1 1872.51
    84.1  1871.9    88.1 1870.15    92.1 1869.18   104.1    1869   116.1 1869.56
   120.1 1870.41   124.1 1872.25   140.1 1884.77   144.1 1887.58   148.1  1889.7
   152.1 1891.05   156.1  1891.9   164.1 1892.95   175.1 1895.97   180.1 1896.94
   200.1 1898.57   204.1  1899.8   212.1 1903.29   216.1 1904.49   223.7 1906.02
#Mann= 3 ,-1,0
       0     .12       0    88.1    .045       0   116.1      .1       0
Bank Sta=88.1,116.1
XS Rating Curve= 0 ,0
Exp/Cntr=0.3,0.1

Type RM Length L Ch R = 1 ,2955    ,137.2,134.9,131.9
XS GIS Cut Line= 2
 2190403.9158464661871.1890356732190661.01459085661755.419425599
#Sta/Elev= 30
       0 1879.86    16.8  1878.5    56.2 1876.24    74.9 1874.03    79.2 1873.81
    92.5 1874.13    95.5 1873.85    98.5 1873.16   107.6 1870.05   110.6 1869.33
   131.5 1868.45   140.7 1866.29     145 1865.54   149.4 1865.55     153 1866.32
   160.8 1868.51   165.1 1870.28   171.4 1873.82   180.1 1879.63   184.5 1881.98
   188.9 1883.78   193.3 1884.81   202.1 1887.88   210.4 1889.89     224 1891.92
   237.6 1895.35   245.9 1896.17   248.4 1896.69   272.3 1904.18     282 1907.49
#Mann= 5 ,-1,0
       0      .1       0      10     .12       0     100      .1       0
   140.7    .045       0     153      .1       0
Bank Sta=140.7,153
XS Rating Curve= 0 ,0
Exp/Cntr=0.3,0.1

Type RM Length L Ch R = 1 ,2820    ,200.3,206.9,212.3
XS GIS Cut Line= 4
2190504.90986104661991.2467910132190533.96872005661973.427132882
2190636.95856798661901.2590642642190674.12110134661875.704846229
#Sta/Elev= 30
       0 1871.03    17.9 1869.37    27.3 1868.81    41.6 1868.29    44.5 1868.09
    51.4 1867.21      56 1866.96    64.6 1867.57    73.2 1867.07    80.7 1867.39
    85.6 1867.34    90.3 1866.47    93.3 1865.55   101.9 1863.39   105.2 1862.88
   113.4 1862.65   119.8 1863.21   124.7 1864.24   129.6 1866.21   139.4  1871.9
   149.1 1879.35     154  1882.1   156.3 1883.07   159.3 1884.23   162.2 1885.07
   179.5 1889.44   183.2 1890.68   188.2  1892.7   197.7 1895.16   204.9 1896.44
#Mann= 3 ,-1,0
       0      .1       0   101.9    .045       0   119.8      .1       0
Bank Sta=101.9,119.8
XS Rating Curve= 0 ,0
Exp/Cntr=0.3,0.1

Type RM Length L Ch R = 1 ,2613    ,165.6,172.9,175.2
XS GIS Cut Line= 2
2190461.84576997662138.8684082232190849.80917802662086.700735545
#Sta/Elev= 30
       0 1872.34    14.5 1870.61    22.5 1868.35    26.6 1867.87    54.8 1868.75
      71 1867.62    83.1 1865.54    91.1 1864.89   107.3 1862.12   175.9 1861.81
   204.2 1862.81   208.2 1862.48   226.21859.259   232.4 1858.14   236.4 1858.34
   240.5 1860.15   249.1 1867.49   256.6 1875.73   259.7 1878.57   268.7 1885.18
   276.8 1892.44   280.8 1895.39   284.9  1896.9     301 1899.03   305.1 1901.72
   309.1 1905.27   313.1 1907.25   349.4 1920.64   361.6 1924.61   391.5 1936.18
#Mann= 4 ,-1,0
       0     .08       0      30      .1       0   226.2    .045       0
   240.5      .1       0
Bank Sta=226.2,240.5
XS Rating Curve= 0 ,0
Exp/Cntr=0.3,0.1

Type RM Length L Ch R = 1 ,2440    ,240.7,240.9,244.8
XS GIS Cut Line= 3
2190439.49478097662216.249921327     2190688.246      662273.851
2190835.66740765662307.963508529
#Sta/Elev= 30
       0 1881.72     4.7 1880.29      13 1876.55    25.3 1873.08    45.9 1868.59
    62.3 1863.41    70.5 1860.06    81.4  1857.8    95.1 1856.33   103.3 1858.49
   123.9  1859.7     160 1859.75   181.4 1858.35   197.8 1859.67     208 1857.23
   214.7 1856.39   226.5 1856.72   234.8 1858.68   247.81856.704   255.3 1855.52
   264.7 1856.48   271.7 1858.73   279.9 1862.49   308.6 1879.02   337.4 1891.78
   357.9 1899.45   370.2 1900.97   373.7 1902.04   382.5 1906.53   406.6  1916.3
#Mann= 5 ,-1,0
       0     .08       0      60     .06       0     160      .1       0
   247.8    .045       0   264.7      .1       0
Bank Sta=247.8,264.7
XS Rating Curve= 0 ,0
Exp/Cntr=0.3,0.1

Type RM Length L Ch R = 1 ,2200    ,224.7,209.4,197
XS GIS Cut Line= 4
2190417.99471053662337.7328368342190443.70458497662347.881471483
2190590.52149956662405.3904011632190656.14933696662433.130002538
#Sta/Elev= 30
       0 1885.29    10.9 1881.45    20.3 1879.18    36.7 1874.06      41 1872.27
    49.6 1868.06    59.9 1863.82    71.1 1857.42    75.4 1855.46      84 1853.17
    92.6 1852.31     100 1852.23   109.3 1851.85   118.4 1852.44     127 1853.69
   131.2 1854.82     134 1855.04   143.2 1854.68     157 1855.75   169.9 1855.72
   200.1 1858.04   204.5 1858.42   208.8 1859.93   213.2 1860.48   221.9 1859.57
   226.2 1858.94   234.9 1856.99   239.2 1856.71   247.5 1857.38   256.6 1859.79
#Mann= 5 ,-1,0
       0      .1       0   77.64     .06       0     100    .045       0
   118.4     .06       0  185.32      .1       0
Bank Sta=100,118.4
XS Rating Curve= 0 ,0
Exp/Cntr(USF)=0,0
Exp/Cntr=0.3,0.1

Type RM Length L Ch R = 1 ,1990    ,146.7,149.9,153.3
XS GIS Cut Line= 3
2190460.00208444 662647.893941582190551.57885324662575.732163331
 2190638.3845773 662505.24876795
#Sta/Elev= 30
       0 1884.29     5.3 1882.08    15.5 1878.65      22 1875.87    30.2 1873.18
      41  1870.1    50.5 1866.73    61.9 1861.79    81.9  1851.2    86.8 1849.75
    91.9 1849.21    94.9 1849.26      97    1849   101.7  1849.9   107.2 1849.79
   112.3  1847.2   114.3 1846.22   118.8 1845.73   122.5  1845.9   127.4 1846.87
   133.3 1849.23   148.3 1851.96     153 1853.21   158.6 1855.09   168.9 1856.49
   184.1 1859.18   187.1 1859.34     207 1859.05   220.4 1859.52   228.4 1860.19
#Mann= 5 ,-1,0
       0     .08       0      40     .06       0   112.3    .045       0
   127.4     .06       0  166.59      .1       0
Bank Sta=112.3,127.4
XS Rating Curve= 0 ,0
Exp/Cntr=0.3,0.1

Type RM Length L Ch R = 1 ,1840    ,164.5,170.1,175.9
XS GIS Cut Line= 3
2190522.84310483662754.249538207     2190644.508      662691.669
2190731.07805282662644.493933851
#Sta/Elev= 30
       0 1865.26    10.5 1861.51    19.5 1857.29    28.5 1852.57      42 1846.61
    46.5 1845.91    52.3 1845.91    64.5 1847.42      87 1846.81      96 1846.25
   109.5 1846.29     116  1845.8   127.4 1843.82   135.4 1842.94     141 1842.87
   149.8 1843.06   153.1 1843.82   154.7 1844.37     159 1846.75   163.8 1847.88
   168.3 1848.21   191.1  1848.2   200.3 1849.36   204.8 1850.55   209.2 1852.27
   213.9 1854.73   218.4 1857.64   223.9 1860.82   227.5 1862.25   235.4 1863.65
#Mann= 5 ,-1,0
       0      .1       0      80     .06       0   127.4    .045       0
   153.1     .06       0  186.82      .1       0
Bank Sta=127.4,153.1
XS Rating Curve= 0 ,0
Exp/Cntr=0.3,0.1

Type RM Length L Ch R = 1 ,1670    ,199.1,187.3,173.8
XS GIS Cut Line= 3
2190542.08792313662855.4351844152190595.53739895662845.963125409
2190779.56597393662839.197368976
#Sta/Elev= 30
       0 1868.33     2.1 1867.22     6.2 1865.74    10.2 1864.87    14.3  1863.5
    17.5 1861.78    58.9 1842.28    62.9 1840.53    70.9 1837.83      75 1837.59
    82.9 1838.49    86.9 1838.49     111 1837.22     119 1837.46     127 1839.18
     129 1839.35     139 1839.33     143 1839.06     147  1839.3     155  1841.1
     167 1842.42     175 1844.08     179 1844.61     191 1845.06     203 1846.73
     211 1847.06     219 1847.89     223 1847.95   233.2  1847.2   238.4 1847.58
#Mann= 5 ,-1,0
       0      .1       0      50     .06       0     139    .045       0
     147     .06       0  154.28      .1       0
Bank Sta=139,147
XS Rating Curve= 0 ,0
Exp/Cntr=0.3,0.1

Type RM Length L Ch R = 1 ,1483    ,143.4,142.7,140.2
XS GIS Cut Line= 2
2190615.98225055663112.8362023132190809.77581922662927.529943227
#Sta/Elev= 30
       0 1865.79     5.8 1863.82    16.9  1863.5    22.7 1862.94    28.2 1860.46
    39.5 1854.69    56.5 1849.47    74.7 1840.86    81.9 1838.74    90.4 1836.91
   109.5 1830.18     121 1828.01     130 1825.78   138.5 1824.97   144.2 1824.91
   152.7 1825.07   158.3 1825.99   169.6 1829.62   178.9 1833.86   182.9 1835.12
   186.6 1835.82   197.9 1836.78   212.1 1837.27   227.2 1838.79   232.7 1839.64
   243.8 1839.88   254.5 1839.29   257.3  1839.4   260.2 1839.67   268.1 1841.28
#Mann= 4 ,-1,0
       0     .06       0     100      .1       0     130    .045       0
   158.3      .1       0
Bank Sta=130,158.3
XS Rating Curve= 0 ,0
Exp/Cntr=0.3,0.1

Type RM Length L Ch R = 1 ,1340    ,112.8,113.5,113.1
XS GIS Cut Line= 2
2190759.32759058663178.4398660152190900.60310214663021.696232757
#Sta/Elev= 30
       0  1833.6     1.7 1833.23    18.5 1831.68    21.3 1831.18    25.2 1830.18
    31.1 1829.17    37.1 1828.86    52.5 1828.83      73 1827.19    78.9 1826.44
    82.5 1825.54    86.5 1823.41    90.9 1820.73    92.1 1820.22    98.6 1818.62
     104 1818.06   108.8 1817.91   120.2    1818   123.3 1818.46   125.6 1818.86
   136.3 1822.67   143.1 1824.24   163.2 1830.29   182.8 1835.41   188.4 1837.55
   190.2 1838.06   194.1  1838.6   202.6 1838.88   206.3 1839.18     211 1840.87
#Mann= 3 ,-1,0
       0      .1       0    98.6    .045       0   123.3      .1       0
Bank Sta=98.6,123.3
XS Rating Curve= 0 ,0
Exp/Cntr=0.3,0.1

Type RM Length L Ch R = 1 ,1227    ,176.1,179.8,183.4
XS GIS Cut Line= 4
2190843.99584057663250.7443320192190857.69621475663236.697008643
2190950.82977553663133.9577442892190976.50001929663111.370090311
#Sta/Elev= 30
       0 1828.17     7.8 1827.76    13.4 1827.25    18.9 1826.39    24.4 1825.84
    32.4 1826.49    41.2  1826.9    51.4 1826.88    56.8 1826.44    60.7 1825.89
    67.6 1824.66      71 1823.72      73 1822.96    74.8 1821.93    80.5 1818.06
    83.3 1816.53    88.8 1814.72    91.8 1814.17    94.7 1813.89   100.7 1814.46
   110.8 1814.16   112.6 1814.35   114.5 1814.79   121.6 1817.23   134.3 1818.94
   145.6 1821.25   154.3 1823.71   165.5 1826.21     174 1828.83   192.5  1833.6
#Mann= 3 ,-1,0
       0      .1       0    91.8    .045       0   112.6      .1       0
Bank Sta=91.8,112.6
XS Rating Curve= 0 ,0
Exp/Cntr=0.3,0.1

Type RM Length L Ch R = 1 ,1047    ,161.6,158.2,157.8
XS GIS Cut Line= 3
2190954.72692964663346.0492978972191093.42442092663263.037044755
2191121.78264404663250.146943336
#Sta/Elev= 30
       0 1820.46     7.5 1819.74    16.3 1818.19    20.3 1817.33    30.9 1816.07
    45.4 1813.65    48.4 1813.31    57.6 1813.16    62.9 1812.73      67 1812.68
    71.7 1812.26    76.3 1811.28    80.9 1809.98    83.3 1809.57    85.6 1809.25
    87.4 1809.24    95.2 1809.54    97.9  1809.2   104.2 1807.38   108.9 1806.82
   113.6 1806.75   118.2 1806.78   121.3 1807.32     130  1809.1   147.5 1811.51
   160.2 1813.07   166.1 1814.07   169.1 1814.87   173.5 1816.61   192.8 1825.73
#Mann= 3 ,-1,0
       0      .1       0   104.2    .045       0   121.3      .1       0
Bank Sta=104.2,121.3
XS Rating Curve= 0 ,0
Exp/Cntr=0.3,0.1

Type RM Length L Ch R = 1 ,889     ,267,252,239
XS GIS Cut Line= 3
2191013.98047776663493.8778550022191119.63525747663406.559855242
2191179.66078634663352.720681929
#Sta/Elev= 30
       0 1815.24    13.7 1814.49    19.1  1814.5    23.6 1814.83    28.8 1814.95
    38.8 1813.07    41.8  1812.3    50.4 1809.84    61.7 1805.96    65.1 1805.04
    70.3 1804.05    80.7 1802.85    82.7 1802.63    91.1 1802.36    95.3 1802.46
    97.61803.064   101.4 1804.42   104.3 1805.09   106.6 1805.48   111.8 1805.81
   121.4  1806.1   132.7 1806.15   139.1 1806.34   157.1 1806.06   164.7 1806.34
   169.1    1807   183.7 1809.94   193.1 1811.47   200.7 1813.19   217.7 1816.24
#Mann= 4 ,-1,0
       0     .06       0      80      .1       0    80.7    .045       0
    97.6      .1       0
Bank Sta=80.7,97.6
XS Rating Curve= 0 ,0
Exp/Cntr=0.3,0.1

Type RM Length L Ch R = 1 ,637     ,105.3,107.6,110.8
XS GIS Cut Line= 3
2191324.58397989663543.7618403212191322.11786167663510.715856176
2191301.89569227663376.559025018
#Sta/Elev= 30
       0 1798.01     6.5 1797.97    10.6 1798.12      14 1798.12    18.6 1797.86
    26.7 1798.14    30.7 1798.04    38.7  1798.1    42.8 1797.93    54.9 1797.17
    67.8 1795.97    71.1 1795.75    75.1 1795.17    80.3 1793.51    83.2 1792.48
    87.3 1792.14    95.4 1792.51    99.4 1793.15   103.5 1794.31   111.6 1798.39
   115.6 1799.34   119.6 1799.69   123.7  1799.9   127.9 1800.31   132.7 1801.19
   139.9 1802.77     148 1805.34     156  1808.5   160.1 1809.95   168.8 1813.77
#Mann= 4 ,-1,0
       0     .05       0      10      .1       0    80.3    .045       0
    99.4      .1       0
Bank Sta=80.3,99.4
XS Rating Curve= 0 ,0
Exp/Cntr=0.3,0.1

Type RM Length L Ch R = 1 ,529     ,105.5,110.7,114.5
XS GIS Cut Line= 4
2191398.35169886663530.4096200012191418.57386826663489.965281196
2191422.51965741663422.3936419732191424.49255199663350.382989955
#Sta/Elev= 30
       0 1797.34    17.2  1796.4    20.2 1796.33    29.1 1796.41    30.9 1796.34
    39.9 1795.76      50 1795.29      62 1794.39    74.1 1792.74    77.8 1792.47
    86.1 1792.12    90.1 1792.57    96.7 1794.02   102.1  1795.1     108 1796.17
   114.1 1797.14   118.1 1798.39   122.1 1801.03   123.5 1802.05   127.4 1805.05
   128.9 1806.32   131.3 1808.16   134.1 1810.45   138.1  1813.3   142.1 1815.29
   162.1 1821.82   170.2  1823.8   178.1 1825.61   182.4 1826.95   184.9 1828.03
#Mann= 4 ,-1,0
       0     .06       0    77.8    .045       0    90.1     .06       0
   95.22      .1       0
Bank Sta=77.8,90.1
XS Rating Curve= 0 ,0
Exp/Cntr(USF)=0,0
Exp/Cntr=0.3,0.1

Type RM Length L Ch R = 1 ,419     ,103.8,118.7,136.1
XS GIS Cut Line= 5
2191369.71251916663578.4308459072191506.01803763663495.250464596
2191515.42661546 663469.79986062 2191537.3476663663397.947527302
2191585.45219454663350.451917143
#Sta/Elev= 30
       0 1798.16    59.1 1797.69    91.9 1795.99   101.6 1796.14   125.3 1795.23
   148.2 1795.06   165.9  1793.6   183.2 1792.91   191.6 1792.93   195.8  1792.5
   199.91790.865   204.2  1789.2   208.4 1788.91   216.8 1789.34   222.7 1790.62
   229.3 1792.98   230.5 1793.85   233.5 1796.24   239.2 1801.47     246 1808.22
   250.2 1811.67   257.9 1816.19   261.9 1817.95   265.9  1819.2   270.1 1820.01
   278.6 1820.23   285.8 1820.99   295.6 1821.46   314.3 1823.28   329.5 1823.68
#Mann= 6 ,-1,0
       0     .05       0      10     .07       0      70     .06       0
   199.9    .045       0   222.7      .1       0  311.94     .03       0
Bank Sta=199.9,222.7
XS Rating Curve= 0 ,0
Exp/Cntr(USF)=0,0
Exp/Cntr=0.3,0.1
